HEC-RAS study SUGARCK.prj: SUGARCK

--- SUGARCK.g01 (geometry) --- (continued)

Type RM Length L Ch R = 1 ,11693   ,157.5,157.5,157.5
XS GIS Cut Line= 3
2196094.42420738588691.2897542222195952.06034014588667.321800904
2195676.42546517588826.700950616
#Sta/Elev= 30
       0 2804.59    10.4 2798.44    30.7 2793.76    42.8 2785.88    52.4 2784.17
    75.3 2775.66    79.4 2771.74    83.4 2766.36    91.5 2762.93   115.9 2761.51
   132.1 2762.28   144.4 2756.41   162.7 2755.64     172 2756.62   210.1 2756.47
   230.5 2753.63   264.4 2751.18   306.7  2755.5   319.8  2751.3   338.3 2752.29
   362.3  2749.4  375.052742.656   382.8 2741.71  393.442742.655   398.4 2745.31
     403 2749.44   409.1 2758.07   435.5 2789.67   443.7 2797.23   462.8 2809.82
#Mann= 5 ,-1,0
       0      .1       0  194.37     .06       0  304.37      .1       0
  375.05    .045       0  393.44      .1       0
Bank Sta=375.05,393.44
XS Rating Curve= 0 ,0
Exp/Cntr=0.3,0.1

Type RM Length L Ch R = 1 ,11536   ,103.6,103.6,103.6
XS GIS Cut Line= 3
2196066.19002949588608.683980185 2195787.8062518588547.171417409
2195600.90269567588712.782163345
#Sta/Elev= 30
       0 2792.31     6.2 2788.78    14.4  2781.2    22.5 2777.58    55.3 2773.69
    75.1  2759.3    79.9 2757.54   100.4 2757.68     125    2761   141.3 2757.62
   198.7 2757.12   231.5 2753.77   247.9 2750.61   291.9 2750.98   300.4 2748.49
   327.4 2749.45   345.8 2746.01   362.8 2746.73   375.5 2749.45   386.1 2746.91
   413.8 2746.75   428.9 2739.14   438.9 2738.01  451.19 2739.13   455.6 2741.55
   466.3 2751.37   487.7 2776.06   511.3 2790.98   519.8 2797.83   534.8 2801.57
#Mann= 5 ,-1,0
       0      .1       0     260     .06       0   428.9    .045       0
  451.19     .06       0   515.1      .1       0
Bank Sta=428.9,451.19
XS Rating Curve= 0 ,0
Exp/Cntr(USF)=0,0
Exp/Cntr=0.3,0.1

Type RM Length L Ch R = 1 ,11432   ,149.1,149.1,149.1
XS GIS Cut Line= 3
2195695.53740763588268.7876397152195686.86255904588469.097780038
2195549.64222669588643.383374572
#Sta/Elev= 30
       0 2773.74    32.4 2763.52    40.4 2760.12    52.4 2752.82    60.4 2750.92
    88.5 2749.89   101.5 2753.12   104.5 2752.97   112.5 2750.09   116.5 2749.83
   128.5 2750.65   140.5 2749.23   197.8 2748.53     221  2747.1   231.1 2744.22
   253.7 2744.35   265.1 2743.01   273.7  2744.5   282.2  2744.3   292.2 2745.73
   301.8 2743.39   307.9 2743.22   314.8  2740.6  327.19 2737.52   343.1  2736.6
   354.92737.518   358.4 2739.01   368.6  2745.2   398.8 2772.74   422.3 2786.72
#Mann= 5 ,-1,0
       0      .1       0     140     .06       0   310.5      .1       0
  327.19    .045       0   354.9      .1       0
Bank Sta=327.19,354.9
XS Rating Curve= 0 ,0
Exp/Cntr(USF)=0,0
Exp/Cntr=0.3,0.1

Type RM Length L Ch R = 1 ,11283   ,128.1,128.1,128.1
XS GIS Cut Line= 3
2195656.48407648588268.7266472082195645.39902204588312.693655654
2195428.26933539588548.324014546
#Sta/Elev= 30
       0  2768.7     8.7 2765.91    25.2 2761.54    29.3 2760.04    37.6 2756.02
    41.7 2753.17      46 2749.47    51.4 2748.03    63.5 2749.21    73.2 2749.58
    84.1 2747.32     106 2744.97   123.9 2744.13   147.5 2742.23   165.2 2741.53
   214.6 2741.29   236.4 2742.69   270.2 2739.02     273 2738.11  281.782733.792
   284.3 2733.01   290.8 2732.78  306.912733.792   318.7  2737.1     324 2739.37
   330.5 2746.78   342.3 2757.53   348.2 2761.84     360 2772.18   365.8  2775.9
#Mann= 4 ,-1,0
       0      .1       0  165.34     .06       0  281.78    .045       0
  306.91      .1       0
Bank Sta=281.78,306.91
XS Rating Curve= 0 ,0
Exp/Cntr=0.3,0.1

Type RM Length L Ch R = 1 ,11155   ,101.3,101.3,101.3
XS GIS Cut Line= 6
2195597.92585571588239.9281744412195467.20770732588414.617213956
2195325.01572971588422.6873325232195292.10223035588410.069019749
2195271.88601047588422.090861826   2195257.50492588452.790382591
#Sta/Elev= 30
       0 2769.49     2.9 2768.37     6.6 2766.21    13.6  2761.3    19.3 2759.08
      25 2758.12    36.3 2758.67    42.2 2757.34      45 2755.53    56.4 2746.07
    62.2 2743.47    91.5 2743.12   101.5  2744.6   107.9  2744.9   116.4 2743.28
   176.4 2738.78   196.4 2738.17   211.4 2736.86   265.5 2735.22   277.3 2733.93
   288.22731.733   321.3 2730.96   338.82731.737   361.5 2733.99   410.1 2733.06
   423.1 2734.31   428.5 2735.77   433.8 2738.07   445.9 2745.81   453.6 2752.08
#Mann= 5 ,-1,0
       0      .1       0     130     .06       0  268.18      .1       0
   288.2    .045       0   338.8      .1       0
#XS Ineff= 1 ,-1
364.3968   453.3    2740
Permanent Ineff=
       F
Bank Sta=288.2,338.8
XS Rating Curve= 0 ,0
Exp/Cntr=0.3,0.1

Type RM Length L Ch R = 1 ,11054   ,258.8,258.8,258.8
XS GIS Cut Line= 3
2195470.09818068588147.6248202192195246.20425563 588413.47902427
2195237.05395367588452.810279351
#Sta/Elev= 30
       0 2764.28    13.8  2759.7    47.9 2758.11    53.6 2757.19    59.6  2754.6
      70 2747.81      82    2741    85.7 2739.34    90.9 2738.06   107.5 2737.99
   127.5 2735.21   148.5 2736.43   167.1 2734.93   184.2 2736.07   201.2 2734.74
   226.5 2736.09   229.6 2735.17  238.262730.052   243.8 2729.26   263.5  2729.1
  270.532730.051   280.7 2731.91   286.3 2734.66   289.2  2735.4   310.6 2733.39
   340.3 2733.05   351.4 2734.21   363.7 2737.34   367.8 2739.34     388 2756.42
#Mann= 5 ,-1,0
       0      .1       0     200     .06       0  238.26    .045       0
  270.53     .06       0     330      .1       0
Bank Sta=238.26,270.53
XS Rating Curve= 0 ,0
Exp/Cntr(USF)=0,0
Exp/Cntr=0.3,0.1

Type RM Length L Ch R = 1 ,10795   ,243.6,243.6,243.6
XS GIS Cut Line= 3
2195254.95109797588031.1901620162194995.79834504588287.031417021
2194965.20919648 588337.73741548
#Sta/Elev= 30
       0 2763.88    19.9  2759.7    31.7 2758.78    65.6 2752.41    82.5 2750.22
    99.6 2746.67   119.3 2740.68   144.4 2730.91   156.1 2727.02   162.3 2726.56
   175.9 2727.65   191.32723.926   196.4 2723.21   209.8 2723.14  217.342723.926
   236.3 2729.41   251.2  2730.5     259 2728.95   273.7 2729.65   293.2 2727.64
   298.9 2728.17   308.8 2730.28   317.3 2727.98   331.5 2726.17   361.5 2726.26
   366.7  2727.2     376 2730.23   403.3 2732.65   408.7  2737.2   423.4 2747.09
#Mann= 5 ,-1,0
       0      .1       0   191.3    .045       0  217.34      .1       0
     320     .06       0  384.16      .1       0
#XS Ineff= 2 , 0
                        305.4575            2735
Permanent Ineff=
       F       F
Bank Sta=191.3,217.34
XS Rating Curve= 0 ,0
Exp/Cntr=0.3,0.1

Type RM Length L Ch R = 1 ,10551   ,206.6,206.6,206.6
XS GIS Cut Line= 4
2195045.40547813587868.5310493692194997.12083167587957.868543157
2194715.58634048588168.0608765422194706.74668328588196.647605501
#Sta/Elev= 30
       0 2770.86      28 2758.32    46.2 2751.19    78.3 2741.67    91.7 2738.69
   100.8 2735.27   104.6 2732.56   112.7  2723.9     116  2721.2  123.682718.169
     136 2716.93   142.7 2717.04  147.742718.166   157.6  2721.9   162.6 2722.88
   198.9 2722.51   244.6 2723.37   274.2 2721.93   287.6 2720.44   342.3 2719.71
   362.3 2722.42   387.5 2719.47   416.1 2720.28   434.7 2719.37   454.1 2720.71
   458.3 2721.82   462.4 2724.45   470.8 2731.85     478 2737.08   482.8 2741.75
#Mann= 4 ,-1,0
       0      .1       0  123.68    .045       0  147.74      .1       0
  351.55     .06       0
#XS Ineff= 2 , 0
                        235.8285            2728
Permanent Ineff=
       F       F
Bank Sta=123.68,147.74
XS Rating Curve= 0 ,0
Exp/Cntr=0.3,0.1

Type RM Length L Ch R = 1 ,10345   ,129,129,129
XS GIS Cut Line= 4
2194937.46130682 587748.669788012194856.58975246587791.834246826
2194745.47078569587988.1470004462194616.23413974588127.411658147
#Sta/Elev= 30
       0 2769.54    18.1 2760.49    33.2  2755.2    43.6 2750.21      69 2731.87
    78.2 2727.12    92.5 2717.62   116.2 2715.43     125 2716.05  129.522713.844
   134.6 2712.71  150.362713.844   157.5 2716.28   165.6 2716.03   180.5 2717.62
   214.3  2717.6   230.6  2716.1   254.1 2719.11   295.5 2718.75   313.8  2720.4
   345.9 2717.18   384.1 2717.72   407.4 2719.97     425 2716.56   444.2 2716.48
   457.6 2717.63   476.9 2716.86   483.1 2719.16   494.4  2729.9   507.2 2738.38
#Mann= 5 ,-1,0
       0      .1       0  129.52    .045       0  150.36      .1       0
  337.25     .06       0  487.25      .1       0
#XS Ineff= 2 , 0
                          157.53            2725
Permanent Ineff=
       F       F
Bank Sta=129.52,150.36
XS Rating Curve= 0 ,0
Exp/Cntr=0.3,0.1

Type RM Length L Ch R = 1 ,10216   ,198.4,198.4,198.4
XS GIS Cut Line= 2
2194860.03474796587638.2315133992194490.26655893587969.112641955
#Sta/Elev= 30
       0 2768.89    15.9 2759.72    40.4 2749.02    58.9 2743.99    69.6 2739.74
     104  2720.8   112.5 2715.14     121 2713.15   142.4 2712.36  151.152710.093
   160.8 2709.04  173.242710.093   178.4 2712.65   183.3 2713.56   200.3 2714.24
   230.6 2712.52   262.4 2715.52   279.6  2713.9   359.4 2715.17   370.3 2713.86
   394.3 2713.58   401.4 2712.34   407.8 2713.32   429.7 2713.35     440    2718
   448.3 2720.11   456.1  2720.8   482.9 2729.24   489.2 2729.83496.1964 2732.37
#Mann= 5 ,-1,0
       0      .1       0  151.15    .045       0  173.24      .1       0
     310     .06       0     440      .1       0
#XS Ineff= 2 , 0
                           198.4            2720
Permanent Ineff=
       F       F
Bank Sta=151.15,173.24
XS Rating Curve= 0 ,0
Exp/Cntr(USF)=0,0
Exp/Cntr=0.3,0.1

Type RM Length L Ch R = 1 ,10017   ,305.2,305.2,305.2
XS GIS Cut Line= 2
 2194802.5870445587532.3253250612194365.71957251587666.087471854
#Sta/Elev= 30
       0 2763.32    10.9 2757.28      25 2746.14    40.2 2735.71    56.6 2720.91
    61.1 2718.03    73.6 2712.58    90.4 2709.95   102.9 2706.35   115.5 2708.19
   136.4 2708.41   149.9 2706.92   165.7 2707.06  175.792704.989   191.6 2705.04
     195 2705.65   203.3 2709.97   207.6 2710.15   224.2 2708.62     241 2708.71
     262 2704.54   289.8 2704.93   299.5 2703.67   320.5    2707   330.8 2705.66
   353.9 2708.15   391.6  2709.1   408.3 2708.26   428.6  2714.2   456.9 2728.43
#Mann= 4 ,-1,0
       0      .1       0  175.79    .045       0   191.6      .1       0
     390     .06       0
#XS Ineff= 2 , 0
                        215.7843            2715
Permanent Ineff=
       F       F
Bank Sta=175.79,191.6
XS Rating Curve= 0 ,0
Exp/Cntr=0.3,0.1

Type RM Length L Ch R = 1 ,9712    ,294.1,294.1,294.1
XS GIS Cut Line= 2
2194611.48319686587266.4497728112194256.58760289587459.247725243
#Sta/Elev= 30
       0 2730.23      28 2720.89    35.6 2716.31    53.8  2702.9   62.53 2698.34
    81.1 2697.75    85.7 2698.34    90.3 2699.54   103.9 2699.46   116.5 2701.08
   131.4 2701.62   151.9 2700.58   176.7  2701.2   185.9 2700.66   196.2 2697.58
   213.2 2697.93   231.4 2701.66     245    2703     264 2703.37   272.3 2702.63
   281.4 2705.04   317.9 2703.87     327  2705.3   340.7 2709.34   345.2 2709.28
   354.3 2707.48   367.3 2708.25   373.2 2709.96   387.9 2719.29   403.9 2722.83
#Mann= 5 ,-1,0
       0      .1       0   62.53    .045       0    85.7      .1       0
     200     .06       0     320      .1       0
#XS Ineff= 2 , 0
                        136.7763            2710
Permanent Ineff=
       F       F
Bank Sta=62.53,85.7
XS Rating Curve= 0 ,0
Exp/Cntr(USF)=0,0
Exp/Cntr=0.3,0.1

Type RM Length L Ch R = 1 ,9418    ,193.4,193.4,193.4
XS GIS Cut Line= 4
 2194529.3717107586997.0098460032194461.81305549587014.399277563
2194241.98085823587173.0101392472194201.88189136 587226.94196482
#Sta/Elev= 30
       0 2722.53      11 2718.86    21.9 2714.16    30.7 2711.98    42.5 2707.52
    67.3 2702.51    71.8 2700.55    78.7 2694.99    84.4 2692.43    90.1 2691.02
    96.4 2690.55   106.3 2689.45  119.88 2690.55   140.8 2694.17   165.5 2693.56
   190.2 2690.02     199 2690.98   214.8  2690.9   227.6 2693.19   239.1  2693.9
   245.4 2694.96   273.5  2695.6   283.9 2696.72   307.9 2694.96   328.3 2695.99
   345.1 2695.95     368 2699.77     388 2707.53   399.4 2709.75     408 2712.43
#Mann= 5 ,-1,0
       0      .1       0    96.4    .045       0  119.88      .1       0
  249.76     .06       0  400.84      .1       0
#XS Ineff= 2 , 0
                        155.6667            2710
Permanent Ineff=
       F       F
Bank Sta=96.4,119.88
XS Rating Curve= 0 ,0
Exp/Cntr=0.3,0.1

Type RM Length L Ch R = 1 ,9225    ,265.9,265.9,265.9
XS GIS Cut Line= 4
2194438.05590082586812.2959700242194376.19601139586821.673331334
2194165.98118503587050.3282574242194100.08440139 587070.36479412
#Sta/Elev= 30
       0 2716.72     5.9 2714.59    22.1 2706.13    38.3 2695.05    54.5 2687.24
    68.5 2686.94    92.1 2689.52   118.9 2690.07   141.5 2688.92   165.1 2689.14
   172.6 2688.09   192.5 2688.63  205.87 2686.94   216.3 2686.06  227.89 2686.94
   239.9 2690.97   274.6 2692.42   281.3 2693.32   287.2 2693.27   304.9 2690.84
   352.2  2693.1   362.3 2692.36   375.1 2692.84   383.4 2695.22   391.8 2698.75
   412.7 2712.09   416.9 2714.18     421 2715.23   425.2 2717.58     442    2733
#Mann= 5 ,-1,0
       0      .1       0  205.87    .045       0  227.89      .1       0
  262.57     .06       0  403.17      .1       0
#XS Ineff= 2 , 0
        119.0651    2695
Permanent Ineff=
       F       F
Bank Sta=205.87,227.89
XS Rating Curve= 0 ,0
Exp/Cntr=0.3,0.1

Type RM Length L Ch R = 1 ,8959    ,236.4,236.4,236.4
XS GIS Cut Line= 4
  2194395.711623586643.8008838772194331.91592492586645.145162495
2194083.03600666586729.454215801 2194016.7841966586774.428672647
#Sta/Elev= 30
       0 2715.67    19.5  2709.3    27.5 2704.21    47.9 2694.08    59.5 2687.16
    66.8 2685.11    85.7 2683.68   127.2 2686.27   164.9 2687.57   169.1 2686.86
   177.6  2682.9   199.3 2683.88   210.2 2682.17   228.2  2681.3   242.2 2682.21
   249.4 2683.38   268.7 2684.63   278.9 2687.63   287.4 2685.57   295.8 2684.91
   312.7  2684.4   321.2 2686.03     330  2685.9     340    2691   354.2  2700.8
   363.9 2705.38   373.6 2708.81   380.3 2712.06   390.2 2715.28   406.7 2722.65
#Mann= 5 ,-1,0
       0      .1       0  163.81     .06       0   210.2    .045       0
   242.2     .06       0  323.81      .1       0
#XS Ineff= 2 , 0
        163.3631    2690   278.9            2691
Permanent Ineff=
       F       F
Bank Sta=210.2,242.2
XS Rating Curve= 0 ,0
Exp/Cntr=0.3,0.1

Type RM Length L Ch R = 1 ,8722    ,332.5,332.5,332.5
XS GIS Cut Line= 4
2194299.41105832586364.4896028852194243.51127615586415.646828152
2193949.77839522586540.7244674952193892.80361249586592.089406372
#Sta/Elev= 30
       0 2722.89     5.6 2719.49    15.2 2709.95    18.8 2707.21    53.7 2686.37
    62.2 2682.17    67.9 2680.29    72.1 2679.59   106.9 2678.57   127.2 2679.47
   135.9 2678.36   149.6 2680.23   192.4    2680   231.6 2681.28  240.892678.214
   259.4 2677.33   270.7 2677.42   275.22678.215   292.9 2680.66   314.2  2680.4
   322.9  2682.8   326.5 2682.98   347.8 2679.82   390.5 2679.23     408 2683.47
   416.3 2688.92   427.6 2695.06   440.3 2698.66   456.4 2706.68   471.7 2713.16
#Mann= 5 ,-1,0
       0      .1       0  240.89    .045       0   275.2      .1       0
  295.77     .06       0  405.03      .1       0
#XS Ineff= 2 , 0
          231.57    2690  324.72            2685
Permanent Ineff=
       F       F
Bank Sta=240.89,275.2
XS Rating Curve= 0 ,0
Exp/Cntr=0.3,0.1

Type RM Length L Ch R = 1 ,8390    ,254.2,254.2,254.2
XS GIS Cut Line= 3
2194120.67766688586092.6013210452193836.82542594586264.427822644
 2193781.2974414586315.558270632
#Sta/Elev= 30
       0 2713.89    14.6 2709.08    29.9 2702.29      38 2696.52    61.4 2675.84
      66  2673.1    80.1 2671.52    94.1 2673.67   122.2 2675.19     126 2674.22
  130.86  2671.3   147.9 2671.31     161 2672.63   190.1 2671.53   201.6 2672.43
   216.3 2670.49     225 2673.15   234.4 2673.28   245.4 2671.02     256 2672.72
   295.2 2675.75   313.9 2675.75   332.9  2677.5   338.1 2678.95   344.1 2682.45
   359.9 2682.64   375.3 2684.51   386.6  2689.3   397.9 2697.26   407.3  2700.3
#Mann= 5 ,-1,0
       0      .1       0  130.86    .045       0   147.9      .1       0
     210     .06       0     320      .1       0
#XS Ineff= 2 , 0
        119.9316    2680
Permanent Ineff=
       F       F
Bank Sta=130.86,147.9
XS Rating Curve= 0 ,0
Exp/Cntr=0.3,0.1

Type RM Length L Ch R = 1 ,8136    ,280.5,280.5,280.5
XS GIS Cut Line= 4
2194054.94066423585944.4197515792193943.39109109586033.474681981
2193750.37640709586015.5506805522193657.66940681586109.524461142
#Sta/Elev= 30
       0 2700.86    34.2 2691.46      68  2687.3    70.8 2685.81      85 2672.32
    90.7 2669.54   110.2 2670.16   121.3 2668.62   136.6 2671.58   142.3 2671.78
     150 2670.44   198.2 2669.87   210.2 2666.06   234.2 2665.29  240.77 2666.04
   246.4  2667.4   258.4 2667.73   266.5 2669.69   274.4    2670   310.7 2667.99
   336.6 2669.59   345.4 2666.94   359.1 2666.06   373.2 2667.73   415.7 2669.38
   430.8 2672.24   436.5  2678.8   460.9 2695.56     465 2697.56   468.6 2697.91
#Mann= 5 ,-1,0
       0      .1       0   210.2    .045       0  240.77      .1       0
  346.58     .06       0  366.58      .1       0
#XS Ineff= 2 , 0
           141.7    2675274.2838            2675
Permanent Ineff=
       F       F
Bank Sta=210.2,240.77
XS Rating Curve= 0 ,0
Exp/Cntr=0.3,0.1

Type RM Length L Ch R = 1 ,7855    ,271.9,271.9,271.9
XS GIS Cut Line= 4
2193987.34194195585799.3493566712193869.44384571585825.706937668
2193620.61430955585835.5413066292193572.62549816585855.742218292
#Sta/Elev= 30
       0 2699.77    11.4 2695.34    22.9 2692.02    27.8 2689.07    44.2 2688.21
    60.6 2682.37    72.9 2680.22    89.3 2676.09   113.9 2667.15     118 2666.37
   146.1 2666.56   154.1 2665.06   170.1 2665.03   190.8 2661.21   206.2 2663.39
   238.2 2661.58   258.2 2662.33  279.61 2660.95   286.2 2659.99   302.2 2660.98
   306.2 2662.76   310.2 2663.19   322.2 2662.71   334.2  2663.4   358.3 2662.42
   374.5 2665.28   383.6 2673.35     392 2679.71     405 2691.91421.8995 2703.09
#Mann= 6 ,-1,0
       0      .1       0  250.81     .06       0  279.61    .045       0
   302.2     .06       0  340.81      .1       0  389.83     .06       0
#XS Ineff= 2 , 0
         207.075    2670 309.769            2670
Permanent Ineff=
       F       F
Bank Sta=279.61,302.2
XS Rating Curve= 0 ,0
Exp/Cntr=0.3,0.1

Type RM Length L Ch R = 1 ,7583    ,280.6,280.6,280.6
XS GIS Cut Line= 4
2193973.67910942 585597.74999532  2193862.045496585594.124781452
2193516.86659382585610.673771546 2193460.9167404 585636.75717742
#Sta/Elev= 30
       0 2705.12     5.5 2701.61    17.5 2700.12      33 2693.26    69.5 2680.23
    89.6 2671.48   105.6 2662.56   112.6  2659.8   133.6 2657.03   149.6 2657.84
  156.572656.008   181.6 2655.98   201.7 2656.13   213.7 2654.62   233.7 2657.47
   249.7 2657.17   257.7 2658.24   265.7 2656.83   293.8 2656.27   305.8 2658.38
   321.8 2656.33   385.9 2657.14   413.9 2661.84   434.3  2658.9     458 2661.22
   462.4  2662.5   466.9 2665.61   480.1 2677.86   493.3 2691.64     519 2711.62
#Mann= 5 ,-1,0
       0      .1       0  156.57    .045       0   181.6      .1       0
  231.69     .06       0  331.69      .1       0
#XS Ineff= 1 ,-1
 257.427 518.999    2670
Permanent Ineff=
       F
Bank Sta=156.57,181.6
XS Rating Curve= 0 ,0
Exp/Cntr=0.3,0.1

Type RM Length L Ch R = 1 ,7303    ,370.8,370.8,370.8
XS GIS Cut Line= 4
2193945.85379218585377.4421238922193869.69229179585322.194185565
2193639.96255439585337.2199399642193602.81014734585307.655489009
#Sta/Elev= 30
       0 2686.91    21.8 2683.67    47.2 2682.99    51.5 2681.31    71.3 2664.06
    87.3 2651.98      91  2649.7    95.6 2648.81   115.7 2648.65   123.7 2647.68
   131.7 2647.39   135.7 2647.56   143.7 2649.47   163.8 2649.76   175.8 2651.15
   195.8 2650.65   211.9 2651.38   218.7 2649.92   227.9 2649.38  240.08 2649.91
   247.9 2651.55     284 2650.61     296 2652.02   308.1 2651.35   320.1 2652.15
   324.4 2652.81   343.6 2660.37   354.7 2664.25   362.9 2665.52371.7906 2668.37
#Mann= 3 ,-1,0
       0      .1       0   218.7    .045       0  240.08     .06       0
#XS Ineff= 2 , 0
                          247.94            2655
Permanent Ineff=
       F       F
Bank Sta=218.7,240.08
XS Rating Curve= 0 ,0
Exp/Cntr=0.3,0.1

Type RM Length L Ch R = 1 ,6932    ,318.8,318.8,318.8
XS GIS Cut Line= 4
2193993.60655972585129.1102335912193921.60293566585131.902610462
2193795.03635489585188.9990228032193585.29844334585181.107263612
#Sta/Elev= 30
       0 2703.03    13.4 2698.76    21.4 2697.19    69.5 2680.43    75.2 2676.42
    86.8 2666.35    98.3 2654.77   104.3 2647.81   108.7 2644.49   110.4 2643.96
   113.1 2643.16   131.6 2642.96   140.6    2644   146.7 2646.18   170.2 2648.07
   209.7 2648.23   225.8 2649.28   237.8 2648.62   257.8 2651.05   288.9 2648.24
   321.8 2648.54   325.8 2649.14   333.9 2653.16   345.9    2652   357.9 2652.75
   361.9 2653.61   365.9 2655.77   373.9 2663.21   381.9 2669.04   420.8 2680.72
#Mann= 5 ,-1,0
       0      .1       0   110.4    .045       0   140.6      .1       0
  260.91     .06       0  360.91      .1       0
Bank Sta=110.4,140.6
XS Rating Curve= 0 ,0
Exp/Cntr=0.3,0.1

Type RM Length L Ch R = 1 ,6613    ,113.6,113.6,113.6
XS GIS Cut Line= 2
2193943.13743874584836.7152381022193545.92847799584853.391950195
#Sta/Elev= 30
       0 2685.03      19  2681.8      34 2672.42      51 2665.23      67 2659.89
      95 2644.46   103.1 2643.59     107 2641.29  112.59 2639.16   139.1 2638.41
  149.31 2639.09   159.1 2642.67   171.1 2642.65   195.1 2640.03   219.2 2640.12
   227.2 2639.61   235.2 2640.53   255.2 2640.88   267.2 2639.18   275.2 2638.79
   279.2    2639   287.2 2640.92   295.2 2641.34   315.2 2640.11   327.3 2640.71
   335.3 2643.93   343.3 2648.25   367.3 2664.19   374.5 2669.59397.5589 2684.06
#Mann= 5 ,-1,0
       0      .1       0     100     .06       0  112.59    .045       0
  149.31     .06       0     200      .1       0
#XS Ineff= 2 , 0
                          171.11            2646
Permanent Ineff=
       F       F
Bank Sta=112.59,149.31
XS Rating Curve= 0 ,0
Exp/Cntr(USF)=0,0
Exp/Cntr=0.3,0.1

Type RM Length L Ch R = 1 ,6500    ,88.3,88.3,88.3
XS GIS Cut Line= 6
2193921.69065411584649.6245342922193824.45224724584652.131049199
2193803.80288403584715.2508135372193762.62581714584777.952256309
 2193747.8451218584832.7458305522193543.23040392 584840.34376999
#Sta/Elev= 30
       0 2673.31     9.5 2674.48    25.5 2673.35    37.5 2667.29    45.5 2664.31
    57.5 2655.81    61.5 2653.88    85.5 2646.86    97.3 2642.28   117.3  2641.4
  156.872637.016   187.9 2636.25  215.082637.015   228.6 2638.46     276 2639.93
   327.1 2639.34   335.1 2640.55   355.2 2640.42   363.2 2641.15   375.2 2638.72
   380.5  2638.6   387.2  2639.1   395.2 2640.83   423.2 2639.75   427.2 2640.18
   446.1 2651.65   467.2 2667.21   475.2 2670.02     490  2680.9   500.2  2685.2
#Mann= 7 ,-1,0
       0      .1       0      80     .06       0  107.27      .1       0
  156.87    .045       0  215.08      .1       0  223.68     .06       0
  295.45      .1       0
#XS Ineff= 2 , 0
                        362.3636            2643
Permanent Ineff=
       F       F
Bank Sta=156.87,215.08
XS Rating Curve= 0 ,0
Exp/Cntr=0.3,0.1

Type RM Length L Ch R = 1 ,6411    ,324.7,324.7,324.7
XS GIS Cut Line= 3
2193922.14342333584643.373494276 2193614.2894999584651.394605404
 2193551.1881747584687.930776176
#Sta/Elev= 30
       0  2672.9      26 2673.37      46 2664.84      54 2658.88      66 2653.28
      82 2647.93      94 2642.97      98 2641.96     126 2641.64     130 2640.38
     134 2637.24  137.262635.684     142 2635.09   162.9 2635.65     170 2637.22
     194 2637.36     206 2638.23     222 2636.22   229.9 2636.66   246.1 2635.82
   254.1 2637.22   298.1 2634.72   310.4  2635.5   313.7 2636.82   324.3  2642.8
   335.5 2650.57   343.5 2654.42   356.6  2663.4   370.5 2670.34   380.9 2674.24
#Mann= 5 ,-1,0
       0      .1       0      80     .06       0  137.26    .045       0
   162.9     .06       0     180      .1       0
#XS Ineff= 2 , 0
                        202.4975            2643
Permanent Ineff=
       F       F
Bank Sta=137.26,162.9
XS Rating Curve= 0 ,0
Exp/Cntr=0.3,0.1

Type RM Length L Ch R = 1 ,6087    ,363.9,363.9,363.9
XS GIS Cut Line= 5
2193773.57578268584219.7969160622193758.34817292584300.474037377
2193691.66732368584390.8964890092193585.32658704584498.921131187
2193508.58726265584515.618723194
#Sta/Elev= 30
       0  2649.3     9.5  2648.4    21.8 2644.64    66.5  2641.4    74.7 2641.79
    87.9 2638.37    92.9  2638.6    97.9 2637.48   102.9 2633.45  107.52 2631.78
   122.7 2631.75   178.6 2634.89   225.7 2632.68   242.6 2633.14   262.2 2631.94
   276.2 2632.58     285  2630.8   294.7 2631.21   304.3 2629.84   320.2 2631.18
   330.6 2630.06   343.6 2630.03   355.4 2631.19   359.5 2633.87   367.7 2641.21
   375.9 2646.45   389.2 2659.87   396.3 2665.69   412.7 2675.92   424.6 2681.96
#Mann= 3 ,-1,0
       0      .1       0  107.52    .045       0   122.7      .1       0
#XS Ineff= 2 , 0
                        187.9819            2643
Permanent Ineff=
       F       F
Bank Sta=107.52,122.7
XS Rating Curve= 0 ,0
Exp/Cntr=0.3,0.1

Type RM Length L Ch R = 1 ,5723    ,295.7,295.7,295.7
XS GIS Cut Line= 5
2193773.10478874584169.354618415 2193645.8690558584191.390619348
 2193504.7036347 584264.783075692193419.58459576584263.612044225
2193365.98136863584288.623741997
#Sta/Elev= 30
       0 2648.88    62.9 2645.26    86.2 2643.07    94.3 2641.65   110.6 2634.98
     131 2631.32   144.6 2629.85   158.4 2629.16   170.3 2630.82   189.6  2630.7
   212.2 2629.13   256.3 2629.27   275.3 2627.55   288.8 2629.67   300.8 2627.68
   320.8 2627.55   324.8 2627.12     3312625.324   336.8    2624   348.8 2623.62
  351.422625.326   352.8 2626.13   360.8 2640.88   368.8 2650.75   372.8 2654.94
   380.1 2659.33   390.4 2662.89   405.4 2673.78   421.3 2681.42432.5125 2688.13
#Mann= 3 ,-1,0
       0      .1       0     331    .045       0  351.42      .1       0
#XS Ineff= 2 , 0
        288.6885    2635
Permanent Ineff=
       F       F
Bank Sta=331,351.42
XS Rating Curve= 0 ,0
Exp/Cntr=0.3,0.1

Type RM Length L Ch R = 1 ,5427    ,275.8,275.8,275.8
XS GIS Cut Line= 4
2193743.72446237583874.3689243522193616.12053993583988.693455056
2193335.84877553583991.8049602452193293.34419713584001.354248888
#Sta/Elev= 30
       0 2654.01    15.8  2653.8    34.2 2649.68    44.2 2646.36    90.7 2641.37
   109.3 2636.52     115 2635.72   143.3 2634.25   155.1 2634.44   171.3 2632.76
   195.3 2632.22   211.3 2630.56   223.3  2630.5   255.3 2627.22   295.3 2625.97
   310.2 2622.92   323.3 2621.59   339.3 2624.03   367.3 2624.47  393.752620.015
   411.3 2618.28  418.152620.016   431.3  2623.6   443.3 2623.36   447.3  2624.3
   463.6 2632.65   475.9 2637.01     480  2639.2   484.1 2640.56495.1799 2641.28
#Mann= 4 ,-1,0
       0     .06       0     130      .1       0  393.75    .045       0
  418.15      .1       0
#XS Ineff= 2 , 0
        359.8427    2625
Permanent Ineff=
       F       F
Bank Sta=393.75,418.15
XS Rating Curve= 0 ,0
Exp/Cntr=0.3,0.1

Type RM Length L Ch R = 1 ,5151    ,334.3,334.3,334.3
XS GIS Cut Line= 4
2193618.51681348 583588.837314142193502.02662601583688.378775872
2193206.79196486583763.5612105062193154.71530154583810.912101407
#Sta/Elev= 30
       0 2683.71    30.3 2672.72    50.1 2663.53    68.3 2658.05    78.5 2650.33
      87 2648.92   101.2 2649.13   105.2 2648.01   113.6 2641.16   134.6 2631.88
   149.4  2623.3   159.3 2622.66   171.6 2619.21   192.3 2617.62   200.5 2617.72
   208.8 2619.24   258.3 2619.63   262.5 2618.86   266.3 2616.35     279    2615
   302.4 2616.35   307.9 2615.91   316.1 2617.45   340.9 2618.78   349.1 2617.85
   369.8 2621.42   398.9 2619.83   466.8 2620.62   515.5 2630.03   528.3 2634.36
#Mann= 4 ,-1,0
       0     .06       0     140      .1       0   266.3    .045       0
   302.4      .1       0
#XS Ineff= 2 , 0
           258.3    2625
Permanent Ineff=
       F       F
Bank Sta=266.3,302.4
XS Rating Curve= 0 ,0
Exp/Cntr=0.3,0.1

Type RM Length L Ch R = 1 ,4817    ,249.5,249.5,249.5
XS GIS Cut Line= 3
2193420.01212593583230.0142801662193068.12907572583626.120479745
2193038.14134777583690.586405798
#Sta/Elev= 30
       0 2734.88     7.8 2731.47    13.5 2725.32    17.8 2722.64    29.9 2721.38
    36.3 2717.93    52.4 2715.81    79.1 2700.19    95.6 2694.25   116.6 2683.37
   127.3 2680.96   138.1 2673.43   152.3 2666.79   163.6 2655.74   186.3 2654.42
   198.5 2641.67   218.2 2627.78   223.6 2623.17   228.8  2616.4  235.872612.163
   257.1 2611.03  265.662612.163   279.8 2613.56     311 2613.28   367.1 2617.18
   378.8 2616.07   512.5 2615.03   559.7 2620.05   586.3 2626.99   600.9  2632.8
#Mann= 4 ,-1,0
       0      .1       0     100     .06       0  235.87    .045       0
  265.66      .1       0
#XS Ineff= 2 , 0
                        361.9419            2620
Permanent Ineff=
       F       F
Bank Sta=235.87,265.66
XS Rating Curve= 0 ,0
Exp/Cntr=0.3,0.1

Type RM Length L Ch R = 1 ,4567    ,325.4,325.4,325.4
XS GIS Cut Line= 3
2193161.81302473583137.3669170742192914.96703067 583515.96541448
2192880.61969688583586.490985502
#Sta/Elev= 30
       0 2691.82    23.7 2682.43    33.2 2680.07    52.3 2670.76    61.7  2667.9
    73.3 2662.24      82 2654.93    99.3 2654.82   102.2 2653.77   110.9 2646.43
   123.9  2637.8   138.3 2621.87   148.5 2612.45   154.2 2608.98     160 2607.97
   190.8 2610.13   205.1 2609.14   226.5 2610.33     241 2608.34   255.4 2607.26
  263.63 2608.28   276.7 2612.55   339.2 2612.78   381.8 2610.95   414.4 2611.86
   453.3 2609.79   481.9 2614.36   499.8 2620.73   511.8 2621.28   530.4 2628.43
#Mann= 5 ,-1,0
       0      .1       0      10     .06       0     190      .1       0
     241    .045       0  263.63      .1       0
#XS Ineff= 2 , 0
                        337.0208            2620
Permanent Ineff=
       F       F
Bank Sta=241,263.63
XS Rating Curve= 0 ,0
Exp/Cntr=0.3,0.1

Type RM Length L Ch R = 1 ,4242    ,336.8,336.8,336.8
XS GIS Cut Line= 4
2192959.72379307582988.8408116612192861.54596443583035.824853237
2192730.03788599583357.6548278322192673.06824713583505.711425259
#Sta/Elev= 30
       0 2659.24     8.4 2658.57    11.9 2657.16    21.7 2649.65    39.4 2648.06
    52.7 2639.91    70.5 2639.44    83.9 2633.59    97.1 2629.78   140.6 2622.23
   149.2 2621.88   163.1 2617.72   175.1 2609.78  197.232604.513   218.2 2603.35
  232.322604.514   270.2 2606.79   300.4 2604.99   313.4 2608.47   339.3 2609.14
   391.2 2604.96     443 2608.59     486 2605.98   520.3 2605.58   528.8 2607.21
   554.6 2608.58     576  2611.6   588.9 2616.79   601.7 2618.19   615.1 2623.15
#Mann= 4 ,-1,0
       0     .06       0  108.84      .1       0  197.23    .045       0
  232.32      .1       0
#XS Ineff= 2 , 0
                        339.4264            2620
Permanent Ineff=
       F       F
Bank Sta=197.23,232.32
XS Rating Curve= 0 ,0
Exp/Cntr=0.3,0.1

Type RM Length L Ch R = 1 ,3905    ,256.8,256.8,256.8
XS GIS Cut Line= 4
2192577.04971472582831.1955692352192548.79337683583115.785621217
2192505.40794977583188.8719224492192425.60081935583418.562311296
#Sta/Elev= 30
       0 2676.53    34.2 2662.28    46.2 2652.84    66.3 2651.97    70.3  2649.8
    82.4 2636.98    98.5 2624.08   106.5 2613.89   126.6 2602.32   146.7 2601.41
   239.2 2603.21   275.3 2600.88   283.4 2602.58  322.592598.568   334.1 2597.28
     3512598.568   357.4 2602.58     362 2603.69   378.5  2603.3   396.7 2599.31
   422.1 2599.93   430.6  2603.6   439.1 2604.16   485.6 2604.17   532.2 2600.69
   574.6 2600.72   578.8 2601.63     600 2612.94   608.4 2613.58   614.1 2615.58
#Mann= 4 ,-1,0
       0     .06       0      90      .1       0  322.59    .045       0
     351      .1       0
#XS Ineff= 2 , 0
                         375.415            2620
Permanent Ineff=
       F       F
Bank Sta=322.59,351
XS Rating Curve= 0 ,0
Exp/Cntr=0.3,0.1

Type RM Length L Ch R = 1 ,3648    ,239.9,239.9,239.9
XS GIS Cut Line= 5
 2192424.2641317582818.2195882042192420.59535694582826.075027238
2192289.57975418 583051.141966312192201.53874913583202.428720859
2192201.68398007583345.117223612
#Sta/Elev= 30
       0 2678.37     9.5 2674.57    17.1 2667.49    21.5 2665.42    34.7 2665.34
    49.3 2662.78    53.9 2660.41    67.8 2649.67    86.3 2638.73   104.9 2620.54
   114.1 2614.55   128.8 2602.33   137.2 2598.17   168.5 2597.22   192.4 2599.92
     216 2597.92   243.7 2598.22  249.852594.967   262.8 2593.53   275.72594.968
   287.8 2597.83   322.4 2597.43   377.9  2599.2     401 2598.31   414.9 2596.03
   446.9 2596.22   462.9 2600.62   502.9 2607.86   518.9 2608.02   586.8 2621.22
#Mann= 4 ,-1,0
       0     .06       0  108.67      .1       0  249.85    .045       0
   275.7      .1       0
#XS Ineff= 2 , 0
          192.38    2605 300.234            2620
Permanent Ineff=
       F       F
Bank Sta=249.85,275.7
XS Rating Curve= 0 ,0
Exp/Cntr=0.3,0.1

Type RM Length L Ch R = 1 ,3409    ,191.2,191.2,191.2
XS GIS Cut Line= 3
 2192191.8252634582746.8042024512192121.20155791582869.914841945
 2191903.7619533583260.643214687
#Sta/Elev= 30
       0 2682.28     7.3 2674.28    30.4  2672.4    42.5 2663.49    62.7 2652.42
    67.3 2647.61    81.1 2645.21    86.5 2642.22     104 2630.72   141.1 2595.99
   145.7 2594.14   159.4  2593.7  167.18 2590.91     189 2589.88  198.072590.908
   206.8 2595.24   223.5 2593.39   237.2 2595.19   259.2 2592.52     283 2593.28
     298 2591.22   324.2  2591.4   379.1 2595.32   397.4 2593.77   475.3  2593.8
   492.1 2599.25   507.3 2599.67   553.9 2615.45   574.5 2624.79   589.1 2625.66
#Mann= 4 ,-1,0
       0     .06       0      50      .1       0  167.18    .045       0
  198.07      .1       0
#XS Ineff= 2 , 0
                           206.8            2600
Permanent Ineff=
       F       F
Bank Sta=167.18,198.07
XS Rating Curve= 0 ,0
Exp/Cntr=0.3,0.1

Type RM Length L Ch R = 1 ,3217    ,212,212,212
XS GIS Cut Line= 3
2192026.96745102582667.1160890512191775.83890789583073.588205322
2191738.38452859583208.669573268
#Sta/Elev= 30
       0 2672.59     2.4 2670.45     5.3 2669.61    25.9 2668.69    35.3 2661.82
    52.9 2652.57    58.8  2647.5      73 2644.92    82.4 2637.05   127.1 2612.46
   134.7 2605.47     143 2596.13   148.2 2591.78   172.1 2589.74  186.342587.042
   209.3  2586.2     2402587.043   286.9 2590.48   303.3 2587.93   345.7 2587.33
   373.9  2590.7   392.7 2590.41     435 2592.27   465.6 2591.74   518.9 2595.04
   527.2 2596.66   547.9 2603.54   568.7 2605.66   589.4 2614.88617.9697 2616.06
#Mann= 4 ,-1,0
       0     .06       0      30      .1       0  186.34    .045       0
     240      .1       0
#XS Ineff= 2 , 0
                          286.89            2600
Permanent Ineff=
       F       F
Bank Sta=186.34,240
XS Rating Curve= 0 ,0
Exp/Cntr(USF)=0,0
Exp/Cntr=0.3,0.1

Type RM Length L Ch R = 1 ,3005    ,281.9,281.9,281.9
XS GIS Cut Line= 4
2191961.56466444582580.5750433642191839.46884114582648.365099338
2191438.46527115582937.267438204 2191402.3780268582946.362594692
#Sta/Elev= 30
       0 2666.11     1.6 2665.12    19.9 2664.09    24.5 2662.19    42.7  2651.3
    51.9 2648.28    60.3 2642.51    72.1 2640.84    88.5 2631.49   120.5 2595.56
   129.7 2592.57   138.8 2586.26   143.7 2585.03   154.7  2584.9  163.692582.005
   183.2 2580.85  193.492582.003   197.9 2584.88   217.7 2586.75   237.4 2584.51
   387.4 2588.67   435.3 2586.56   524.2 2588.13   577.6 2586.99   583.9 2589.35
   598.2    2599     617  2607.9   648.6 2608.47     661 2616.11   671.1 2619.53
#Mann= 3 ,-1,0
       0      .1       0  163.69    .045       0  193.49      .1       0
#XS Ineff= 2 , 0
                        220.9684            2590
Permanent Ineff=
       F       F
Bank Sta=163.69,193.49
XS Rating Curve= 0 ,0
Exp/Cntr=0.3,0.1

Type RM Length L Ch R = 1 ,2724    ,237.6,237.6,237.6
XS GIS Cut Line= 4
 2191878.1966916582365.5219083812191750.10613833582399.476767131
2191399.69164993 582509.120286232191303.02282309582507.120094363
#Sta/Elev= 30
       0 2653.83     2.1 2651.91     6.2  2650.5    22.8 2649.76    35.2 2642.56
    60.3 2632.59    72.4 2624.51    84.9 2622.93   113.8 2595.27   123.5  2587.3
   134.5 2581.04   155.5 2579.61  174.332576.076   193.2 2574.85  204.632576.075
   214.2 2581.64   243.5 2582.45   281.2 2580.26   306.4 2581.64   448.9 2576.64
   461.5 2577.32   478.2 2576.38   486.7 2577.53   499.7 2576.57   511.2 2579.87
   523.2 2588.62     536 2596.24   579.2 2615.69   591.2 2622.08   596.4 2626.29
#Mann= 4 ,-1,0
       0     .06       0     110      .1       0  174.33    .045       0
  204.63      .1       0
#XS Ineff= 2 , 0
                        299.8367            2585
Permanent Ineff=
       F       F
Bank Sta=174.33,204.63
XS Rating Curve= 0 ,0
Exp/Cntr=0.3,0.1

Type RM Length L Ch R = 1 ,2486    ,244,244,244
XS GIS Cut Line= 4
2191839.88690091582141.8625343352191648.51903968582172.494396412
2191384.50992638582315.6772555262191280.61081425 582324.36524965
#Sta/Elev= 30
       0 2639.22     3.8 2637.39      24 2636.32    36.2 2628.55    68.6 2615.02
    84.8 2610.59   103.9 2602.69   109.1 2598.99   124.9 2596.05   133.4 2591.98
   173.8 2583.95   194.2 2578.01   221.5 2576.42  233.572572.755   247.7 2571.57
   266.22572.755   280.7  2581.3   294.3 2576.95   317.1 2575.66   339.8 2576.82
   389.3 2574.34   418.8 2576.04     449 2575.79     463 2573.41   498.5 2574.07
   502.5  2575.4   514.4 2583.98   542.6 2606.34   578.8 2621.81   598.4 2632.37
#Mann= 4 ,-1,0
       0     .06       0      60      .1       0  233.57    .045       0
   266.2      .1       0
#XS Ineff= 2 , 0
                        283.2046            2585
Permanent Ineff=
       F       F
Bank Sta=233.57,266.2
XS Rating Curve= 0 ,0
Exp/Cntr=0.3,0.1

Type RM Length L Ch R = 1 ,2242    ,304.5,304.5,304.5
XS GIS Cut Line= 4
2191830.75616956581818.1620622242191522.87334519581841.477684877
2191393.39001897582133.3157548012191263.79400936582153.287855432
#Sta/Elev= 30
       0  2633.5    14.6 2626.36    22.6 2618.85    42.7  2617.3    66.8 2604.63
    83.5 2600.88   126.9 2587.21   183.1 2576.41   203.2 2569.93   247.3 2570.86
   339.1 2569.71   448.5 2574.75   483.5  2574.4   487.9 2573.62   495.5 2569.19
   514.1 2568.39  521.45 2569.15   531.6 2571.51   592.9 2573.59   619.1 2571.41
   633.3 2572.54   646.5 2570.26   657.6 2571.03   673.8 2583.53   681.9 2586.34
   702.1 2600.15   718.3 2606.79   730.7 2614.57   746.6 2628.32   759.2 2633.66
#Mann= 5 ,-1,0
       0      .1       0      60     .06       0     150      .1       0
   495.5    .045       0  521.45      .1       0
#XS Ineff= 2 , 0
        449.7087    2575597.5739            2585
Permanent Ineff=
       F       F
Bank Sta=495.5,521.45
XS Rating Curve= 0 ,0
Exp/Cntr=0.3,0.1

Type RM Length L Ch R = 1 ,1937    ,310.4,310.4,310.4
XS GIS Cut Line= 4
2191822.23847397581630.3713525742191425.37598635581787.222006834
2191243.12825816581798.9766677642191201.06511248581825.100231724
#Sta/Elev= 30
       0 2634.53    15.1 2629.62      28 2622.92    49.5 2619.02    66.7 2610.77
    75.3 2603.31   101.1 2602.67     114 2595.93     160 2582.78   200.1 2573.98
   234.5  2571.6   389.1 2566.85   431.9 2570.48     448 2568.54     456 2565.91
   488.1 2568.27   492.1 2567.67  497.642563.846   508.1 2562.59  518.592563.844
   524.1 2565.35   552.2 2567.28   564.2 2578.88   572.8 2585.05   584.3 2596.38
   592.3  2601.8     616 2623.39   633.4 2625.52     648 2634.55658.8756 2639.25
#Mann= 5 ,-1,0
       0      .1       0      50     .06       0     160      .1       0
  497.64    .045       0  518.59      .1       0
#XS Ineff= 2 , 0
           488.1    2575
Permanent Ineff=
       F       F
Bank Sta=497.64,518.59
XS Rating Curve= 0 ,0
Exp/Cntr=0.3,0.1

Type RM Length L Ch R = 1 ,1627    ,417,417,417
XS GIS Cut Line= 4
2191667.85210927581319.4649446512191520.44143886581419.148870323
2191177.73554721581522.6929930462191099.99374338581635.553658362
#Sta/Elev= 30
       0 2606.56    12.5 2604.28    60.2 2590.87   116.2 2585.11   130.6 2576.61
   147.9 2574.71   163.8 2565.74   176.7 2562.87     220 2561.17   232.6 2563.21
   270.2 2563.43   291.1 2562.08   366.3 2564.06   392.4 2561.06   423.7 2560.48
   430.1 2557.87   437.3 2556.73   458.2 2557.77   470.7 2561.51   479.1 2565.93
   508.3 2567.03   516.7 2571.79   529.2 2576.65   568.1  2587.2   579.1 2592.44
   593.5 2594.18   607.9  2601.9     628 2609.71   645.8 2618.29673.0032 2628.48
#Mann= 4 ,-1,0
       0     .06       0     170      .1       0   430.1    .045       0
   458.2      .1       0
#XS Ineff= 2 , 0
           410.8    2566
Permanent Ineff=
       F       F
Bank Sta=430.1,458.2
XS Rating Curve= 0 ,0
Exp/Cntr=0.3,0.1

Type RM Length L Ch R = 1 ,1210    ,343.8,343.8,343.8
XS GIS Cut Line= 4
2191328.59233269580891.9758473062191094.88977724581133.621987404
2190993.81254014 581239.57275671 2190865.0808736581312.171400854
#Sta/Elev= 30
       0 2590.78    12.8 2585.01    23.9 2576.58    40.6 2567.14    52.4 2555.85
    58.1 2552.83   139.8 2555.46   165.2 2554.67   179.4 2556.86   230.8 2555.92
   252.9 2557.56   268.8 2556.71   279.9 2553.33   307.7  2557.2   329.3  2556.1
  337.752551.375   346.6 2550.47  371.872551.374   385.3 2557.19   405.7 2555.05
   414.2 2556.94   422.7 2555.84   457.2 2557.36   487.9 2576.01   548.8 2595.98
   573.1 2605.74   585.5 2613.24   608.5 2623.84   620.1 2631.64   630.4    2632
#Mann= 5 ,-1,0
       0      .1       0      60     .06       0     200      .1       0
  337.75    .045       0  371.87      .1       0
#XS Ineff= 2 , 0
        310.9396    2558
Permanent Ineff=
       F       F
Bank Sta=337.75,371.87
XS Rating Curve= 0 ,0
Exp/Cntr=0.3,0.1

Type RM Length L Ch R = 1 ,866     ,225.6,225.6,225.6
XS GIS Cut Line= 4
 2191235.7005444580769.0618145362191012.15501891580951.042882531
2190836.13357054580962.2688239312190739.69053015581034.300724276
#Sta/Elev= 30
       0 2594.57    14.9 2588.85    38.2  2576.8      51 2568.78    65.1 2556.57
    81.9 2549.89   102.1 2552.22   167.5 2552.21   179.9 2555.07   190.2 2552.97
     213 2552.78   226.3 2550.07   240.9 2552.89   261.3 2551.24   292.2 2552.55
   332.3 2548.78   345.9 2551.98   396.5 2553.16   404.5 2552.99   408.5 2551.24
  415.612544.854   429.7  2543.7  449.932544.852   464.6 2550.15   474.6 2551.69
   484.6 2563.49   499.5 2572.88   556.4 2592.22   575.3 2603.06585.0057 2603.64
#Mann= 5 ,-1,0
       0      .1       0      90     .06       0     190      .1       0
  415.61    .045       0  449.93      .1       0
Bank Sta=415.61,449.93
XS Rating Curve= 0 ,0
Exp/Cntr=0.3,0.1

Type RM Length L Ch R = 1 ,641     ,316.1,316.1,316.1
XS GIS Cut Line= 2
2191137.93521583580550.3158781432190609.72491325580862.655802568
#Sta/Elev= 30
       0 2604.67      16 2594.26    29.2 2590.41      81  2569.1   108.9 2548.79
   131.4 2547.29     160 2547.96   169.8 2545.71   181.5 2546.48   192.6 2549.48
   211.2 2550.25   215.8 2549.73   225.1  2544.4   229.7 2544.24   243.7 2545.96
   322.7  2548.3   333.4 2546.14   356.7 2546.97  371.692541.827   391.8 2540.65
  407.282541.828   415.6 2547.53   447.2 2546.12   453.6 2547.21   470.6 2554.04
   508.6 2562.34   555.3  2574.7   573.6 2580.99   590.3 2591.35613.6468 2593.08
#Mann= 5 ,-1,0
       0      .1       0     150     .06       0     290      .1       0
  371.69    .045       0  407.28      .1       0
#XS Ineff= 2 , 0
           322.7    2552
Permanent Ineff=
       F       F
Bank Sta=371.69,407.28
XS Rating Curve= 0 ,0
Exp/Cntr(USF)=0,0
Exp/Cntr=0.3,0.1

Type RM Length L Ch R = 1 ,324     ,,,
XS GIS Cut Line= 2
2191053.64922686580297.0152327312190453.25753573580644.268805437
#Sta/Elev= 30
       0  2604.3    10.9 2602.39    20.2 2597.05    38.7 2592.86    80.2 2577.02
   103.4 2574.78   117.2  2570.8   136.1 2555.46   153.4 2545.36   269.7 2543.43
   273.5 2542.35  279.25 2537.37     294 2536.26   305.7 2537.38   325.2 2539.09
   337.9 2537.98   343.7 2539.57   352.9 2537.87   371.4 2543.83   422.2 2542.33
   436.1 2544.42   478.4 2540.67     510 2542.31   523.9 2545.11   557.4 2569.87
   563.3 2572.72   583.9 2574.62   651.1 2573.09   676.3 2577.12693.5814 2574.37
#Mann= 3 ,-1,0
       0      .1       0  279.25    .045       0   305.7      .1       0
Bank Sta=279.25,305.7
XS Rating Curve= 0 ,0
Exp/Cntr(USF)=0,0
Exp/Cntr=0.3,0.1
LCMann Table=0

Chan Stop Cuts=-1
Use User Specified Reach Order=0
Composite Channel Slope=5
